--- DERRICKCK.prj (project) ---

Proj Title=DERRICKCK
Current Plan=p01
Default Exp/Contr=0,0
English Units
Geom File=g01
Flow File=f01
Plan File=p01
BEGIN DESCRIPTION:
END DESCRIPTION:
DSS Export Rating Curves= 0
DSS Export Rating Curve Sorted= 0
DSS Export Volume Flow Curves= 0
DXF OffsetX= 0
DXF OffsetY= 0
DXF ScaleX= 0
DXF ScaleY= 0

--- DERRICKCK.p01 (plan) ---

Plan Title=Floodplain
Program Version=4.00
Geom File=g01
Flow File=f01
K Sum by GR=0
Std Step Tol=0.01
Critical Tol=0.01
Num of Std Step Trials=20
Max Error Tol=0.3
Flow Tol Ratio=0.001
Split Flow NTrial=30
Split Flow Tol=0.02
Split Flow Ratio=0.02
Log Output Level=0
Friction Slope Method=1
Unsteady Friction Slope Method=2
Unsteady Bridges Friction Slope Method=1
Global Log Level=0
CheckData=False
Run HTab=0
Run UNet=0
Run PostProcess=0
UNET Theta=0
UNET Theta Warmup=0
UNET ZTol=0
UNET ZSATol=0
UNET MxIter=0
UNET MaxInSteps=0
UNET DtIC=0
UNET DtMin=0
UNET MaxCRTS=0
UNET WFStab=0
UNET SFStab=0
UNET WFX=0
UNET SFX=0
UNET DSS MLevel=0
UNET DZMax Abort=0
UNET Convert EG Bridges=0
UNET Use Existing IB Tables=0
UNET Froude Limit=0
UNET Froude Power=0
Write IC File=0
Echo Input=False
Echo Output=False
Write Detailed=0

--- DERRICKCK.f01 (steady flow) ---

Flow Title=NFF Regression Equation
Program Version=4.10
Number of Profiles= 1
Profile Names=P100yr
River Rch & RM=DERRICKCK,Main            ,10923.2
895.7978
River Rch & RM=DERRICKCK,Main            ,9509.2
965.3159
River Rch & RM=DERRICKCK,Main            ,7358.3
1138.498
River Rch & RM=DERRICKCK,Main            ,6729.6
1164.481
River Rch & RM=DERRICKCK,Main            ,4865.6
1257.319
River Rch & RM=DERRICKCK,Main            ,3346
1317.946
River Rch & RM=DERRICKCK,Main            ,497.4
1413.897
Boundary for River Rch & Prof#=DERRICKCK,Main            , 1
Up Type= 0
Dn Type= 3
Dn Slope=0.002
DSS Import GetInterval= 0
DSS Import GetPeak= 0
DSS Import FillOption= 0

--- DERRICKCK.g01 (geometry) ---

Geom Title=USGS 10m DEM
Program Version=4.10

River Reach=DERRICKCK       ,Main
Reach XY= 30
     1770641.399      558434.735     1770583.158      557996.721
     1770645.756      557365.989     1770534.645      557169.808
     1770702.613      556901.145     1770733.024      556714.323
     1770901.971      556572.794     1771078.915      556191.509
     1771522.926      555851.666     1771598.447      555769.634
     1771610.166      555609.478     1771788.551      555442.811
     1771901.832      555126.405     1771828.916      554744.895
     1771858.863      554587.343      1772119.28      554181.093
     1772226.079      553431.988     1772519.266      552849.343
     1772736.468      552168.072     1772990.374      551957.134
     1773429.176      552002.707     1773701.311      551898.541
     1773858.864      551684.999     1774292.457       551423.28
     1774671.364      551442.812     1775020.322      551553.488
     1775287.928      551888.151     1775474.749      551746.197
     1775574.908      551934.505     1775835.792      551837.215

Type RM Length L Ch R = 1 ,10923.2 ,48.1,53.6,59
XS GIS Cut Line= 2
     1770767.377       558415.23     1770542.117      558411.324
#Sta/Elev= 26
       0  654.41     9.8  653.91    19.6   653.5    29.4   653.1    39.2  652.68
      49  652.27    58.8  651.77    68.6  651.26    78.4  650.74    88.2  650.23
      98  649.54   107.8  648.56   117.5   647.7   118.6  647.67   127.3  647.42
   133.6  648.42   137.1  648.98   146.9  653.72   156.7  660.06   166.5  666.51
   176.3  673.76   186.1  681.74   195.9   690.2   205.7  698.91   215.5  707.54
   225.3  715.73
#Mann= 3 , 0 , 0
       0      .1       0   117.5    .045       0   133.6      .1       0
Bank Sta=117.5,133.6
XS Rating Curve= 0 ,0
Exp/Cntr=0.3,0.1

Type RM Length L Ch R = 1 ,10869.6 ,38.7,38.8,38.9
XS GIS Cut Line= 2
     1770798.627      558399.605     1770565.554      558338.408
#Sta/Elev= 28
       0  655.28     9.6  654.93    19.3  654.43    28.9  653.91    38.6  653.32
    48.2  652.76    57.8  652.19    67.5  651.61    77.1  651.09    86.8  650.53
    96.4  649.95     106   649.4   115.7  648.83   125.3  648.22     135  647.56
   144.6   647.2   144.8   647.2   154.2  647.41   159.8   648.7   163.9  649.64
   173.5  652.91   183.1  655.89   192.8  659.21   202.4  663.37   212.1  668.36
   221.7  673.95   231.3  679.95     241  686.32
#Mann= 3 , 0 , 0
       0      .1       0   144.8    .045       0   159.8      .1       0
Bank Sta=144.8,159.8
XS Rating Curve= 0 ,0
Exp/Cntr=0.3,0.1

Type RM Length L Ch R = 1 ,10830.8 ,115.6,103.4,91.3
XS GIS Cut Line= 2
     1770815.554      558364.449     1770582.481      558303.251
#Sta/Elev= 28
       0  653.98     9.6  654.88    19.3  654.74    28.9  654.16    38.6  653.53
    48.2  652.97    57.8  652.42    67.5  651.94    77.1  651.43    86.8  650.94
    96.4  650.45     106  649.95   115.7  649.49   125.3  649.03     135  648.48
   144.6   647.8   154.2  647.27   155.5  647.28   163.9  647.32   170.5  647.83
   173.5  648.06   183.1  650.04   192.8  652.63   202.4  655.23   212.1  658.32
   221.7   661.9   231.3  665.81     241  670.02
#Mann= 3 , 0 , 0
       0      .1       0   154.2    .045       0   170.5      .1       0
Bank Sta=154.2,170.5
XS Rating Curve= 0 ,0
Exp/Cntr=0.3,0.1

Type RM Length L Ch R = 1 ,10727.4 ,215.8,216.4,216.9
XS GIS Cut Line= 2
     1770767.377      558186.064     1770560.346      558244.658
#Sta/Elev= 25
       0  653.88     9.8  653.04    19.6   652.3    29.3  651.65    39.1  651.09
    48.9  650.53    58.7  649.96    68.5  649.38    78.2  648.82      88  648.19
    97.8   647.5   107.6  646.78   117.4  646.12   121.2  645.97   127.1  645.74
   136.2  645.87   136.9  645.88   146.7  646.77   156.5  648.92   166.3  652.82
     176     658   185.8   662.9   195.6  667.18   205.4  671.41   215.2  675.38
#Mann= 3 , 0 , 0
       0     .06       0   117.4    .045       0   136.9      .1       0
Bank Sta=117.4,136.9
XS Rating Curve= 0 ,0
Exp/Cntr=0.3,0.1

Type RM Length L Ch R = 1 ,10511   ,236.4,242.2,247.8
XS GIS Cut Line= 2
     1770747.846       557971.22     1770504.356       558033.72
#Sta/Elev= 29
       0  652.72     9.7  651.76    19.3  651.04      29  650.43    38.7  649.91
    48.3  649.43      58  648.95    67.7  648.54    77.4  648.16      87  647.78
    96.7  647.37   106.4  646.95     116  646.54   125.7  646.16   135.4  645.71
     145  645.16   154.7  644.51   157.9  644.41   164.4  644.22   172.9  645.05
     174  645.16   183.7  647.76   193.4  653.67     203  661.43   212.7  669.24
   222.4  676.95     232   684.5   241.7  691.93   251.4  699.46
#Mann= 3 , 0 , 0
       0     .06       0   154.7    .045       0     174      .1       0
Bank Sta=154.7,174
XS Rating Curve= 0 ,0
Exp/Cntr=0.3,0.1

Type RM Length L Ch R = 1 ,10268.8 ,138.2,138.4,138.4
XS GIS Cut Line= 2
     1770749.148      557779.814     1770514.773      557781.116
#Sta/Elev= 28
       0  652.43     9.8  651.93    19.5  651.35    29.3  650.67    39.1  649.98
    48.8   649.2    58.6  648.24    68.4  647.17    78.1  645.92    87.9  644.48
   91.01  644.13    97.7  643.31    98.1   643.3   107.4  643.01   113.1  643.48
   117.2  643.82     127  645.36   136.7  648.18   146.5  652.31   156.2  656.88
     166  661.65   175.8  666.67   185.6  671.86   195.3  677.12   205.1  682.46
   214.8  687.76   224.6  693.02   234.4  698.16
#Mann= 3 , 0 , 0
       0     .06       0   91.01    .045       0   117.2      .1       0
Bank Sta=91.01,117.2
XS Rating Curve= 0 ,0
Exp/Cntr=0.3,0.1

Type RM Length L Ch R = 1 ,10130.5 ,259.1,247.2,234.2
XS GIS Cut Line= 4
     1770859.319      557719.339      1770687.95      557645.699
     1770595.502      557645.699     1770516.075      557676.949
#Sta/Elev= 22
       0  656.15     9.8  655.51    29.4  654.44    39.3  653.77    58.9  652.14
    88.4  651.41    98.2  651.06   157.1  648.31   186.5  647.12   195.8  646.56
   214.3  645.15     242  642.82   251.2  642.34   260.5  642.79   269.7  645.88
   288.4  656.31   297.9   661.3   307.4  666.65   316.9  672.15   335.9  683.69
   354.8  695.62   364.3  701.52
#Mann= 3 , 0 , 0
       0     .06       0     242    .045       0   260.5      .1       0
Bank Sta=242,260.5
XS Rating Curve= 0 ,0
Exp/Cntr=0.3,0.1

Type RM Length L Ch R = 1 ,9883.3  ,121.7,124.8,128.5
XS GIS Cut Line= 4
     1770763.833      557304.409     1770697.065      557373.564
     1770579.877       557433.46     1770508.263      557451.689
#Sta/Elev= 30
       0  679.79     9.6  678.96    19.2  677.67    28.8  674.88    38.4  671.09
    48.1  669.18    57.7  667.16    67.3  663.66    76.9   658.7    86.5  653.48
    96.1  648.59   105.5  645.38   114.9  643.34   124.3  641.97   133.7  640.73
   143.1  639.92   152.5  639.51   161.9  639.72  164.61  640.14   180.7  643.56
   190.1  644.66   208.9  646.09     237  648.83   246.2  650.01   255.4  651.38
   264.7  653.12   273.9  655.17   283.2  657.52   292.4  660.25   301.6  663.41
#Mann= 3 , 0 , 0
       0      .1       0   143.1    .045       0  164.61     .06       0
Bank Sta=143.1,164.61
XS Rating Curve= 0 ,0
Exp/Cntr=0.3,0.1

Type RM Length L Ch R = 1 ,9758.4  ,226.6,249.2,272.4
XS GIS Cut Line= 3
      1770687.95      557251.168     1770462.226      557346.894
     1770241.336       557308.46
#Sta/Elev= 30
       0   665.2    19.6  654.53    29.4  649.61    39.2  646.79    58.8  644.26
    78.5  639.97    88.3  639.28    98.1   640.1   101.4  640.81   117.7  643.78
   176.5  645.89   186.3  647.74   215.8   659.2   254.9   673.5   274.4  681.75
   284.2   686.4   293.9  691.48   303.7   697.3   313.4  703.84   332.9  717.88
   342.7  724.32   352.4  730.07   362.2  735.17   371.9  739.28   381.7  742.25
   391.4  744.35   401.2  745.74   420.6  747.28   449.9  747.97   469.4  747.33
#Mann= 3 , 0 , 0
       0      .1       0    78.5    .045       0   101.4     .07       0
Bank Sta=78.5,101.4
XS Rating Curve= 0 ,0
Exp/Cntr=0.3,0.1

Type RM Length L Ch R = 1 ,9509.2  ,186.5,188.6,190.3
XS GIS Cut Line= 4
     1770707.481      557137.887     1770642.377      557123.564
     1770497.846      557023.303     1770391.075      556885.283
#Sta/Elev= 30
       0  673.55     9.5  668.86      19  665.23    28.6   663.7    38.1  659.83
    57.1  648.69    66.7  644.66    86.2  641.37      96  639.27   104.5  637.84
   105.8  637.62   115.5  637.82   119.5  638.36   135.1  640.23   154.6  640.52
   193.7  640.27   203.5  640.49   213.2   641.1   232.8   642.8   281.3  647.75
   300.7  649.23   320.1  650.27   329.8  651.72   339.5   654.6   349.2  656.94
   358.9  660.11   368.6  667.67   378.3  676.45     388  683.41   417.1  702.56
#Mann= 3 , 0 , 0
       0     .08       0   104.5    .045       0   119.5     .06       0
Bank Sta=104.5,119.5
XS Rating Curve= 0 ,0
Exp/Cntr=0.3,0.1

Type RM Length L Ch R = 1 ,9320.6  ,178.6,151.9,124.5
XS GIS Cut Line= 2
     1770772.586      557007.678      1770562.95      556827.991
#Sta/Elev= 27
       0  670.18     9.5   663.4      19  656.78    28.6  654.56    38.1  651.95
    47.6  648.64    57.1  645.88    66.6   643.9    76.2  642.42    85.7  641.16
    95.2  639.46   104.7  637.06   111.6  635.97   114.2  635.56   123.8  635.68
   126.6  636.47   133.3  638.36   142.8  640.59   152.3   641.6   161.9  641.84
   199.9  642.42   209.5  642.64   228.5  643.15     238  643.53   257.1  644.14
   266.6  645.31   276.1  649.03
#Mann= 3 , 0 , 0
       0     .06       0   111.6    .045       0   126.6     .06       0
Bank Sta=111.6,126.6
XS Rating Curve= 0 ,0
Exp/Cntr=0.3,0.1

Type RM Length L Ch R = 1 ,9168.7  ,157.3,68,61.8
XS GIS Cut Line= 4
     1770896.283      556713.408     1770823.367      556736.845
       1770781.7      556755.074      1770618.94      556827.991
#Sta/Elev= 22
       0  645.21     9.6  644.36    28.7  642.93    57.4  642.21    76.6  641.91
    94.8   641.5   122.1  641.18   150.2  641.03   159.6  640.72     169  639.35
   178.4  636.67  184.77  635.56   187.8  635.02   197.2  634.79   203.8  635.62
   206.6  635.97   215.9  638.26   225.3  640.47   234.7  641.53   262.9  641.61
   272.3  641.74   300.4  642.62
#Mann= 3 , 0 , 0
       0     .06       0  184.77    .045       0   203.8     .06       0
Bank Sta=184.77,203.8
XS Rating Curve= 0 ,0
Exp/Cntr=0.3,0.1

Type RM Length L Ch R = 1 ,9100.8  ,28.1,126.5,155.8
XS GIS Cut Line= 4
     1770880.658      556662.626     1770807.742      556686.064
     1770766.075      556704.293     1770603.315       556777.21
#Sta/Elev= 29
       0  642.43     9.6  642.15    19.2  641.75    28.7  641.04    38.3  640.12
    47.9  639.34    76.6  638.06    85.7  638.05     113  637.65   122.1   637.3
   131.5  637.21   140.8  636.36   150.2  635.65   154.2  635.27   159.6  634.76
     169  634.29   178.4  635.14   187.8   636.9   197.2  639.54   206.6  641.53
   215.9  642.21   234.7  642.96   244.1   643.7   253.5  644.63   262.9  645.68
   272.3  649.85   281.6  655.25     291  658.95   300.4  659.25
#Mann= 3 , 0 , 0
       0      .1       0   154.2    .045       0   178.4     .06       0
Bank Sta=154.2,178.4
XS Rating Curve= 0 ,0
Exp/Cntr=0.3,0.1

Type RM Length L Ch R = 1 ,8974.3  ,29.2,44.1,44.9
XS GIS Cut Line= 6
     1770877.331       556655.61     1770863.442       556659.95
     1770854.832      556665.523     1770818.158      556641.793
     1770760.867      556609.241     1770671.023      556570.178
#Sta/Elev= 29
       0  641.84     7.3  641.81    14.6  641.54    19.7  641.47    24.8  641.08
    33.5  638.57      40  636.36    42.3  635.58      51  633.94      55  634.15
    59.8   634.4    68.5  636.15    77.9  638.38    87.3  640.23    96.7  641.52
   106.1  642.64   115.6  643.35     125  643.66   134.4   644.8   144.2  648.58
     154  654.23   163.8  660.07   173.6  665.51   183.4   671.1   193.2   677.2
     203  683.58   212.8  689.88   222.6  696.19   232.4  702.53
#Mann= 3 , 0 , 0
       0     .08       0      40    .045       0    59.8     .08       0
Bank Sta=40,59.8
XS Rating Curve= 0 ,0
Exp/Cntr=0.3,0.1

Type RM Length L Ch R = 1 ,8930.2  ,337.1,337.2,337.2
XS GIS Cut Line= 5
     1770910.172      556645.699     1770891.943      556639.189
     1770847.672      556610.543     1770790.381      556577.991
     1770700.537      556538.928
#Sta/Elev= 28
       0  640.43     9.7  640.17    19.4  639.53    28.2  638.11    36.9  635.98
    42.5  634.75    45.7  634.04    54.5  633.44    57.5  633.63    63.3  633.99
    72.1  635.27    81.5  636.76    90.9  638.56   100.3  640.11   109.7  641.05
   119.2  641.49   128.6  642.08     138   642.9   147.8  643.78   157.6   646.1
   167.4  650.84   177.2  657.05     187  663.32   196.8   669.5   206.6  675.58
   216.4  682.06   226.2  688.56     236  695.05
#Mann= 3 , 0 , 0
       0     .08       0    42.5    .045       0    63.3     .06       0
Bank Sta=42.5,63.3
XS Rating Curve= 0 ,0
Exp/Cntr=0.3,0.1

Type RM Length L Ch R = 1 ,8593    ,453.5,461.3,468.7
XS GIS Cut Line= 3
     1771127.331      556397.652     1771048.121      556346.654
     1770866.914      556227.296
#Sta/Elev= 21
       0  656.26     9.4  654.46    28.3  650.61    56.5  644.35      66  642.31
   113.1  632.27   121.4  630.63   122.5  630.41   131.9  629.64   141.4  630.21
   150.8  632.17   160.2  634.61   169.7     636     198  639.63   207.4  640.75
   235.7  643.86   254.6  645.74     264  646.77   273.5  647.27   292.3  647.48
   311.2  647.99
#Mann= 3 , 0 , 0
       0     .06       0   121.4    .045       0   141.4     .06       0
Bank Sta=121.4,141.4
XS Rating Curve= 0 ,0
Exp/Cntr=0.3,0.1

Type RM Length L Ch R = 1 ,8131.7  ,127.8,124.7,121.6
XS GIS Cut Line= 4
     1771474.553      556096.003     1771379.067      556074.302
     1771306.367      555978.816     1771223.902      555913.711
#Sta/Elev= 26
       0  647.94    19.6  645.45    29.4   644.1    58.8  640.29    78.3  637.53
    97.9  634.55   116.4   632.7   134.8  631.28   144.1  630.67   153.3  629.83
   162.5  628.78   171.8  627.96     181   627.7   190.2  628.48   199.5  630.79
   208.7  634.79   217.9  639.22   227.5  644.03     237   649.3   246.6  654.97
   256.1  660.98   265.7  667.25   284.8  680.66   303.9  693.93   313.4  700.14
     323     706
#Mann= 3 , 0 , 0
       0     .06       0   171.8    .045       0   190.2      .1       0
Bank Sta=171.8,190.2
XS Rating Curve= 0 ,0
Exp/Cntr=0.3,0.1

Type RM Length L Ch R = 1 ,8007    ,140.7,140.6,140.5
XS GIS Cut Line= 2
      1771520.56      556028.005     1771347.817      555855.262
#Sta/Elev= 28
       0  645.72     9.8  644.29    19.5  642.82    29.3  641.46    39.1   640.1
    48.9  638.69    58.6  637.34    68.4  636.03    78.2  634.69      88  633.42
    97.7  632.07   107.5  630.36   115.1  628.86   117.3  628.42     127  627.71
   130.1  627.96   136.8   628.5   146.6  630.88   156.4  633.25   166.1  635.57
   175.9  638.67   185.7  642.39   195.4  646.35   205.2  650.68     215  655.39
   224.8   660.6   234.5  666.02   244.3  671.55
#Mann= 3 , 0 , 0
       0     .06       0   115.1    .045       0   136.8      .1       0
Bank Sta=115.1,136.8
XS Rating Curve= 0 ,0
Exp/Cntr=0.3,0.1

Type RM Length L Ch R = 1 ,7866.4  ,29.5,29.5,29.5
XS GIS Cut Line= 4
     1771595.213      555982.939     1771561.576      555870.092
     1771484.536      555794.137     1771381.454      555740.968
#Sta/Elev= 27
       0  646.89    19.6   642.9    39.2   639.3    58.9  635.26    68.7  633.81
    78.5  632.97    88.3  632.48   107.9  631.97   117.8  631.64   127.6  631.19
   137.4  630.28   147.3  628.31   157.1  626.86   166.9  627.28  169.88  627.96
   176.8   629.8   186.6  631.75   196.4   632.8   216.1  634.42   225.9   635.7
   235.6  637.91   245.3  642.17   264.6  652.68   274.3  657.84   283.9  662.78
   293.6  667.48   341.9  690.37
#Mann= 3 , 0 , 0
       0     .07       0   147.3    .045       0   166.9     .06       0
Bank Sta=147.3,166.9
XS Rating Curve= 0 ,0
Exp/Cntr=0.3,0.1

Type RM Length L Ch R = 1 ,7836.9  ,62.9,61.6,60.2
XS GIS Cut Line= 4
     1771617.782      555963.842     1771584.145      555850.994
     1771507.105       555775.04     1771404.024      555721.871
#Sta/Elev= 30
       0  646.76     9.8   644.9    19.6  642.79    29.4  639.79    39.2  636.43
    49.1  634.19    58.9  632.98    68.7  632.33    78.5  631.97   107.9  631.28
   127.6  630.71   137.4  630.15   147.3   628.7     156  626.99   157.1  626.77
   166.9  625.96   176.8  628.29   186.6   631.2   196.4  632.46   206.3  633.15
   225.9  634.35   235.6  635.31   245.3  637.17   254.9  640.93   264.6  646.12
   274.3  651.16   293.6  661.37   303.3  666.01   322.6  674.84   341.9  683.97
#Mann= 3 , 0 , 0
       0     .08       0     156    .045       0   176.8     .06       0
Bank Sta=156,176.8
XS Rating Curve= 0 ,0
Exp/Cntr=0.3,0.1

Type RM Length L Ch R = 1 ,7775.3  ,163.7,166.1,167.4
XS GIS Cut Line= 4
     1771723.685      555854.394     1771636.879       555811.86
     1771538.789      555725.922      1771489.31      555593.978
#Sta/Elev= 30
       0   640.9     9.7  639.73    38.7  635.47    48.3  634.21      58  633.19
    67.7  632.49    77.3  631.93     106  630.59   115.3  630.04   124.6  629.33
   133.9  628.47   143.2  627.23   152.6  625.72   161.9  624.94   171.2  625.47
   180.5  627.51   189.8  629.38   199.1  630.36   208.4  630.96   236.5  632.37
   245.9  634.23   255.3  637.28   264.6  640.58   283.4  646.48   302.2  652.26
   311.6  655.42   330.4   662.1   339.8  665.24   349.2  668.22     368  673.93
#Mann= 3 , 0 , 0
       0     .06       0   152.6    .045       0   171.2     .06       0
Bank Sta=152.6,171.2
XS Rating Curve= 0 ,0
Exp/Cntr=0.3,0.1

Type RM Length L Ch R = 1 ,7609.3  ,258.3,251,244.3
XS GIS Cut Line= 3
     1771778.373      555920.222     1771667.695      555673.911
      1771510.36      555512.236
#Sta/Elev= 30
       0  669.19    28.9  656.93    38.6  653.06    48.2  649.46    57.9  646.07
    67.5  643.12    77.2  641.06    86.8  639.48    96.4  638.44   115.7   636.7
     135  635.37   183.2  632.53   202.5  631.56   231.5  630.92   260.4  630.89
   299.5  630.56   309.3  630.03   319.1  628.75   328.9  626.94   338.7  625.48
   348.5  624.44   358.3  624.23   368.1  625.19   377.9  630.65   387.7  644.26
   397.5  652.47   407.4  656.43     476  680.36   485.8   684.1   495.6  688.09
#Mann= 3 , 0 , 0
       0     .08       0   338.7    .045       0   368.1      .1       0
Bank Sta=338.7,368.1
XS Rating Curve= 0 ,0
Exp/Cntr=0.3,0.1

Type RM Length L Ch R = 1 ,7358.3  ,283.2,280.6,277.6
XS GIS Cut Line= 5
     1772112.574      555839.927     1771967.415       555525.71
     1771883.624       555493.79     1771761.011        555427.6
     1771668.781      555365.751
#Sta/Elev= 30
       0  642.66    86.5  644.24   144.2   646.6   163.4   646.8   173.1   646.4
   182.7  645.52   192.3  644.46   201.9  642.96   211.5  642.21   230.8  641.48
   240.4  641.61   259.6  640.84   278.8   639.4   346.1  636.18   435.8  629.77
   454.4  628.82   482.2   627.9   510.1  626.49   519.4  625.66   528.7  624.21
   547.3  623.65   556.6  624.06   565.8  625.67   575.1  628.88   584.4   633.2
   593.6   638.2   612.1  647.29   658.4  668.02   676.9  675.62   686.2  679.69
#Mann= 3 , 0 , 0
       0     .06       0   528.7    .045       0   556.6      .1       0
Bank Sta=528.7,556.6
XS Rating Curve= 0 ,0
Exp/Cntr=0.3,0.1

Type RM Length L Ch R = 1 ,7077.7  ,172.8,159.1,145.4
XS GIS Cut Line= 4
     1772038.789      555229.033     1771963.919      555212.757
     1771871.689      555175.864     1771757.756      555169.354
#Sta/Elev= 20
       0   632.5    19.2  631.36    57.5  629.34   103.7  626.57   112.7  626.11
   130.8   625.4   139.8  624.38   148.9  622.74   157.9  621.75   166.9  622.33
     176  626.58   185.5  633.39     195  640.31   204.5  647.38     214   654.6
   223.5  660.94     233  665.95   242.5  670.15   261.5  678.13   290.1  689.98
#Mann= 3 , 0 , 0
       0     .06       0   148.9    .045       0   166.9      .1       0
Bank Sta=148.9,166.9
XS Rating Curve= 0 ,0
Exp/Cntr=0.3,0.1

Type RM Length L Ch R = 1 ,6918.5  ,188.1,188.9,189.8
XS GIS Cut Line= 3
     1772136.445      554996.828     1772033.364      554993.572
     1771783.798      555052.166
#Sta/Elev= 27
       0  637.19    28.1  633.14    46.9  630.66    56.2  629.64    65.6  628.74
    84.4  627.17   103.1  626.07   122.1  625.24   141.1  624.64   188.6  623.35
   207.6  622.86   217.1  622.74   226.6  622.46   236.1  621.44   245.6  620.28
     255  620.23   257.9  620.98   264.5  622.68     274  628.25   283.5  634.32
     293  639.44     312  650.05   321.5  655.27     331  660.13   340.5  664.64
     350  668.81   359.5  672.76
#Mann= 3 , 0 , 0
       0     .06       0   236.1    .045       0   257.9      .1       0
Bank Sta=236.1,257.9
XS Rating Curve= 0 ,0
Exp/Cntr=0.3,0.1

Type RM Length L Ch R = 1 ,6729.6  ,49.8,49.8,49.8
XS GIS Cut Line= 4
     1772106.064       554877.47     1771915.091      554836.237
     1771884.709      554836.237      1771739.31      554864.449
#Sta/Elev= 27
       0   634.7     9.8  630.74    19.5  628.48    29.3  627.76    39.1  627.24
    48.8  626.86   107.5  625.13   146.5  624.11   175.8  623.41     203  622.88
     235  622.64   244.3  622.26   253.5  620.81   258.4  619.74   262.8  618.77
     272  618.49   281.3  619.55   290.6  623.02   299.8  625.16   309.1  625.83
   318.3  627.03   327.6  630.03   336.8   634.4   346.1  639.43   355.4   644.9
   364.6  650.52   373.9  656.03
#Mann= 3 , 0 , 0
       0     .06       0   258.4    .045       0   281.3      .1       0
Bank Sta=258.4,281.3
XS Rating Curve= 0 ,0
Exp/Cntr=0.3,0.1

Type RM Length L Ch R = 1 ,6679.8  ,138.3,148.7,158.7
XS GIS Cut Line= 4
     1772101.723      554827.557     1771910.751      554786.324
     1771880.369      554786.324      1771734.97      554814.536
#Sta/Elev= 24
       0  640.36     9.8  635.57    19.5  631.06    29.3  627.94    39.1  626.71
   117.2  624.49   166.1  623.42   195.4  622.57   225.8   622.5   244.3   622.7
   253.5  621.46   262.8  619.32     272  618.22   281.3  618.78   290.6  621.14
   299.8  624.52   309.1  626.78   318.3  627.87   327.6   628.7   336.8  630.45
   346.1  634.49   355.4  639.96   364.6  646.01   373.9  652.31
#Mann= 3 , 0 , 0
       0     .06       0   262.8    .045       0   281.3     .08       0
Bank Sta=262.8,281.3
XS Rating Curve= 0 ,0
Exp/Cntr=0.3,0.1

Type RM Length L Ch R = 1 ,6531.1  ,242.8,249.8,256.6
XS GIS Cut Line= 3
     1772086.532      554696.263     1772011.662      554693.008
     1771730.629      554618.138
#Sta/Elev= 28
       0  635.73     9.4  630.57    18.7  627.33    28.1  626.33    46.8  625.78
    65.6  625.02    84.6  624.13    94.3  623.84   113.7  623.55   171.9  623.22
   181.6  623.08   191.3  622.42     201  621.41   210.7  620.96   220.4  620.99
     230  620.39   239.8  618.56   249.4  617.56   259.1  618.38   268.8  621.71
   288.2  631.17   297.9  635.33   307.6  637.89   317.3  639.02     327     640
   336.7  640.89   356.1  642.08   365.8  643.26
#Mann= 3 , 0 , 0
       0     .06       0   239.8    .045       0   259.1     .06       0
Bank Sta=239.8,259.1
XS Rating Curve= 0 ,0
Exp/Cntr=0.3,0.1

Type RM Length L Ch R = 1 ,6281.2  ,328.9,324.5,320.1
XS GIS Cut Line= 4
     1772206.975      554587.757     1772009.492      554461.888
     1771929.197       554410.89     1771859.753      554345.786
#Sta/Elev= 28
       0  673.03     9.8  668.65    29.3  660.22      39  655.63    48.8  649.74
    58.6  643.43    68.3  636.92    78.1  630.62    87.8  625.86    97.6  623.96
   156.1  622.65   234.2  621.38   253.2  620.25   262.7  620.16   272.2  620.18
   281.7  618.65   290.7  617.04   291.3  616.93   300.8  616.67   310.3  618.06
   319.8  620.96   329.3  624.59   338.8  628.34   357.9  636.12   367.4  640.33
   376.9  644.68   395.9  653.97   424.5  667.64
#Mann= 3 , 0 , 0
       0     .06       0   290.7    .045       0   310.3      .1       0
Bank Sta=290.7,310.3
XS Rating Curve= 0 ,0
Exp/Cntr=0.3,0.1

Type RM Length L Ch R = 1 ,5956.7  ,301.5,293,284.5
XS GIS Cut Line= 4
     1772422.904      554294.788     1772305.026      554225.418
     1772096.298      554143.963     1772005.152       554094.05
#Sta/Elev= 24
       0   680.8    58.6  653.25    78.2  643.45   107.5  628.11   117.2  623.27
     127  620.52   136.8  619.98   146.5  619.83   195.2  619.62   234.2  619.58
   273.2  619.31   282.9   619.1   292.6  618.57   302.4  617.86   312.1  616.21
   321.9  613.73   322.4  613.69   331.6  612.89   341.4  614.36   351.1  618.31
   360.8     623   389.2  635.84     427  653.65   464.8  671.11
#Mann= 3 , 0 , 0
       0     .06       0   322.4    .045       0   341.4      .1       0
Bank Sta=322.4,341.4
XS Rating Curve= 0 ,0
Exp/Cntr=0.3,0.1

Type RM Length L Ch R = 1 ,5663.7  ,337.6,341.4,345.2
XS GIS Cut Line= 3
      1772362.14        553865.1     1772140.786      553866.185
     1772032.279      553884.632
#Sta/Elev= 24
       0  620.83    48.1  618.91    96.2  617.17   144.4  615.24     154   614.9
   163.6  614.66   173.2  613.58   182.9  611.53   192.5  610.37   202.1   611.9
   202.6  612.18   211.7  617.29   221.4   625.2   230.5  632.35   248.9   645.1
     258  651.25   267.2  655.88   276.4  658.95   285.6  662.15   294.7  665.64
   303.9  669.75   313.1  674.46   322.2   679.6   331.4  684.91
#Mann= 3 , 0 , 0
       0     .06       0   182.9    .045       0   202.6      .1       0
Bank Sta=182.9,202.6
XS Rating Curve= 0 ,0
Exp/Cntr=0.3,0.1

Type RM Length L Ch R = 1 ,5322.3  ,89.4,93.7,97.9
XS GIS Cut Line= 4
     1772346.949      553582.982     1772236.055      553531.839
     1772177.678      553522.218     1772005.152      553573.217
#Sta/Elev= 28
       0  624.58      47  620.93   103.3  616.74   112.7  616.15   122.1  615.77
   130.6  613.97     139  611.13   147.5  608.77   155.9  608.22   164.4   609.4
   172.8  613.26   181.3  616.21   190.8  617.28   209.7   617.9   219.2  617.94
   228.6  617.39   238.1  616.59   247.6  615.91     257  615.82   266.5  618.14
     276  624.01   294.9  637.13   304.4   643.8   313.8  649.97   323.3  655.25
   332.8  659.93   342.2  664.38   361.2  673.22
#Mann= 3 , 0 , 0
       0     .06       0     139    .045       0   164.4     .06       0
Bank Sta=139,164.4
XS Rating Curve= 0 ,0
Exp/Cntr=0.3,0.1

Type RM Length L Ch R = 1 ,5228.6  ,60.2,60.1,60.2
XS GIS Cut Line= 2
     1772338.268      553476.645     1771936.793      553329.076
#Sta/Elev= 30
       0  620.56    58.3  618.02      68  617.74    77.8  617.93    87.5   618.9
    97.2  617.67   106.9  612.66   112.6   610.4   116.7  608.78   126.4  609.16
   130.2  610.41   145.8  616.25   155.5  616.91   184.7  614.71   194.4  613.79
   204.2  613.36   233.3  613.36   262.5  613.95   281.9  614.11   291.6  614.76
   301.4  616.06   320.8  619.23   340.2  623.01     350  624.13   359.7  624.57
   369.4  624.23   379.1  623.24   398.6  620.53   408.3  618.91   427.7  617.09
#Mann= 3 , 0 , 0
       0     .06       0   112.6    .045       0   130.2     .06       0
#XS Ineff= 2 , 0
                           151.9          618.45
Permanent Ineff=
       F       F
Bank Sta=112.6,130.2
XS Rating Curve= 0 ,0
Exp/Cntr=0.3,0.1

Type RM Length L Ch R = 1 ,5168.4  ,67.9,69.9,71.8
XS GIS Cut Line= 2
     1772371.906      553425.647      1771970.43      553278.078
#Sta/Elev= 30
       0  619.62    19.4  620.08    29.2  620.02      68  618.56    77.8  618.79
    87.5   619.8    97.2   620.2   106.9  617.35   116.7  611.75     119  610.96
   126.4   608.4   136.1  608.92  139.06  611.02   145.8  614.51   155.5  618.28
   165.3  618.79   184.7  618.24   204.2  618.49   213.9     618   233.3  614.71
     243  613.61   252.8  613.18   291.6  612.97   311.1  613.63   320.8  613.68
   359.7  612.84   379.1  613.34   388.8   614.3     418  619.03   427.7   620.2
#Mann= 3 , 0 , 0
       0     .06       0     119    .045       0  139.06     .06       0
#XS Ineff= 2 , 0
                           164.3          620.07
Permanent Ineff=
       F       F
Bank Sta=119,139.06
XS Rating Curve= 0 ,0
Exp/Cntr=0.3,0.1

Type RM Length L Ch R = 1 ,5098.5  ,229.5,232.9,236.1
XS GIS Cut Line= 2
     1772376.246      553362.713     1771994.301      553183.677
#Sta/Elev= 30
       0  624.55     9.8  619.42    19.6  616.67    29.4  616.13    39.2     616
      49  615.36    58.9  614.13    68.7  613.18    78.5   611.9    88.3  609.69
    90.2  609.41    98.1  608.23   107.9  608.53  112.93   609.4   127.5  611.88
   137.3  612.39   186.4  613.45     206  613.66   225.6  613.61   235.4  613.46
   245.2  613.14   264.9  611.83   274.7  611.77   284.5  612.06   294.3     613
   304.1  614.61   313.9  616.04     363  622.88     412  629.58   421.8  631.18
#Mann= 3 , 0 , 0
       0     .08       0    90.2    .045       0  112.93     .06       0
Bank Sta=90.2,112.93
XS Rating Curve= 0 ,0
Exp/Cntr=0.3,0.1

Type RM Length L Ch R = 1 ,4865.6  ,569.8,572.5,573.7
XS GIS Cut Line= 4
     1772471.732      553173.911     1772412.053      553128.338
     1772221.081       553002.47     1772088.702      552953.642
#Sta/Elev= 30
       0  667.02     9.4  659.29    18.8  651.22    28.2  642.98    37.5  634.22
    46.9  629.28    56.3  626.82    65.7  623.55    75.1  619.16    84.6  614.48
    94.2  609.97   100.9  607.82   103.7  606.92   113.2  605.99   122.7  607.12
   132.3  609.31   141.8  610.32   179.9  610.96   227.6  612.03   284.8   613.6
   294.3  613.93   303.8  614.88   313.2  617.03   322.6  619.75     332  622.22
   369.7   629.2   388.5  633.13   397.9  635.43   407.3  638.39   444.9  651.98
#Mann= 3 , 0 , 0
       0      .1       0   100.9    .045       0   122.7     .06       0
Bank Sta=100.9,122.7
XS Rating Curve= 0 ,0
Exp/Cntr=0.3,0.1

Type RM Length L Ch R = 1 ,4293    ,285.3,280.4,276.3
XS GIS Cut Line= 4
     1772794.215      552832.331     1772620.603      552608.373
     1772471.298       552493.79     1772386.228       552377.47
#Sta/Elev= 30
       0  638.77     9.8  635.36    19.5  633.18    39.1  630.52    78.2  626.08
    97.7  624.33   175.9  620.86   224.7  616.76   254.1  615.18   273.6  612.95
   292.8  609.23   311.6  606.54   321.7  604.23   330.4  603.11   339.8  603.01
   349.2  604.19   358.6  607.21   368.1  608.49   424.5  608.75   462.2  610.59
   471.6  611.39   481.2  612.93     510   620.3     558  633.93   567.6  637.03
   577.2  641.12   586.9   646.3   596.5  650.13   606.1  651.78   615.7  652.78
#Mann= 3 , 0 , 0
       0     .06       0   321.7    .045       0   349.2     .06       0
#XS Ineff= 2 , 0
       0                     383       0     620
Permanent Ineff=
       F       F
Bank Sta=321.7,349.2
XS Rating Curve= 0 ,0
Exp/Cntr=0.3,0.1

Type RM Length L Ch R = 1 ,4012.6  ,278.1,285.4,291.7
XS GIS Cut Line= 4
     1772878.199      552465.343     1772754.501      552362.261
     1772621.037      552293.902     1772559.189      552225.542
#Sta/Elev= 29
       0  612.64    47.4  610.74    66.3   610.1    85.2  609.76   142.1  609.29
   151.6  608.94   170.4  607.67   179.8   607.2   189.1  606.94   198.5  606.82
   217.2     607   226.6  606.99   245.4  606.47   254.7  605.94   264.1  604.45
   270.7  603.22   273.5   602.7   282.8  602.23   292.2  603.39   301.6     609
     311   616.1   320.2  622.45   329.4  627.08   338.6  628.84   357.1  631.62
   366.3     634   375.5  637.67   393.9  645.48   403.2   649.2
#Mann= 3 , 0 , 0
       0     .06       0   270.7    .045       0   292.2      .1       0
Bank Sta=270.7,292.2
XS Rating Curve= 0 ,0
Exp/Cntr=0.3,0.1

Type RM Length L Ch R = 1 ,3727.2  ,380.9,381.2,382.8
XS GIS Cut Line= 3
     1773131.454      552390.491     1772790.742       552056.29
     1772623.642      552036.758
#Sta/Elev= 30
       0  629.53    29.2   620.6      39  618.47    58.4  615.26   116.9  610.53
   165.6  608.78   253.2  606.99   311.7  607.07   379.9  608.06   389.6  607.76
   409.1  606.33   418.8  604.56   426.1  602.42   428.6  601.69   438.3  600.79
     448  601.38   457.8  603.63   467.5  607.34     496  621.54   505.3  624.93
   514.6  626.55   533.3   626.9   542.7  627.48   589.4   631.3   598.8  632.36
   608.1  634.39   617.5  638.06   626.8  644.57   636.2  652.76   645.5  659.33
#Mann= 3 , 0 , 0
       0     .06       0   426.1    .045       0   457.8      .1       0
Bank Sta=426.1,457.8
XS Rating Curve= 0 ,0
Exp/Cntr=0.3,0.1

Type RM Length L Ch R = 1 ,3346    ,240.8,241.2,238
XS GIS Cut Line= 3
     1773358.451      552293.269     1773102.374      551883.112
     1772996.037      551752.904
#Sta/Elev= 30
       0  669.88    19.3  658.63      29  654.71    38.7  652.01      58  648.01
    67.7  644.87    77.4   643.3      87  642.66    96.7  640.34   164.4  607.52
   174.1  604.75   222.4  603.73   338.5  603.68   348.1  603.08   367.5  599.64
   386.8  598.72   396.5  599.05   406.2  600.49   415.8  603.25   425.5   604.2
   454.5   605.4   464.2  606.76   483.5  611.56   492.9  612.75   502.2  613.48
   539.6  614.22   586.3  616.11     605  617.64   623.6  619.82   651.6  624.97
#Mann= 3 , 0 , 0
       0      .1       0   367.5    .045       0   396.5     .06       0
Bank Sta=367.5,396.5
XS Rating Curve= 0 ,0
Exp/Cntr=0.3,0.1

Type RM Length L Ch R = 1 ,3104.8  ,110.9,112,115.5
XS GIS Cut Line= 4
     1773566.784       552150.04     1773434.406      552056.724
      1773345.43      551948.217     1773230.412        551687.8
#Sta/Elev= 30
       0  634.82     9.5  634.44      19  635.13    38.1  635.56    57.2  635.35
    76.2  633.18    85.7   631.6    95.3  629.95   104.8  627.02   114.3  622.91
   123.8  617.83   133.4  613.63   142.9  610.67   152.4  609.17     162  608.08
     190  605.57   199.4  603.79   208.7  600.51   218.1  598.32   227.4  597.41
   237.6  598.09   246.2  600.07   264.9   605.3   274.2  606.06   283.6  606.32
   400.4  606.81   488.8  610.62   528.1  611.47   547.7  612.65     587  612.64
#Mann= 3 , 0 , 0
       0     .06       0   218.1    .045       0   237.6     .06       0
Bank Sta=218.1,237.6
XS Rating Curve= 0 ,0
Exp/Cntr=0.3,0.1

Type RM Length L Ch R = 1 ,2992.8  ,26.6,32.6,38
XS GIS Cut Line= 4
       1773660.1      552100.126     1773527.722       552006.81
     1773438.746      551898.303     1773323.728      551637.887
#Sta/Elev= 30
       0  612.74    38.1  610.57    85.7  606.83   104.8  605.67   142.9  604.05
     162  603.58   180.7  602.79     190  602.07   199.4  600.44   208.7  598.03
   218.1  597.16   227.4  597.55   230.9  598.32   236.8  599.62   246.2  602.72
   255.5  604.32   274.2   605.6   283.6  606.38   292.9  607.46   302.3  608.09
   312.1   608.2   341.6  607.77     371  606.42   380.8  606.24   400.4  606.52
   420.1  607.23   449.5  607.79   508.4  610.08   547.7  611.93     587  614.75
#Mann= 3 , 0 , 0
       0     .08       0   208.7    .045       0   230.9     .06       0
Bank Sta=208.7,230.9
XS Rating Curve= 0 ,0
Exp/Cntr=0.3,0.1

Type RM Length L Ch R = 1 ,2960.2  ,37.8,37.7,37.7
XS GIS Cut Line= 4
     1773647.079       552078.28     1773536.836      551985.398
     1773458.711      551817.864     1773428.329      551740.607
#Sta/Elev= 30
       0  610.52    19.2  609.14    28.8  608.31    57.7  605.14    67.3  604.39
    76.9  603.82    96.1   603.1   105.7  602.88   115.3  602.75   144.2  602.71
   153.9  602.41   163.6  601.32   173.3  598.63   183.1  597.24   192.8  597.21
   197.3  598.13   202.5   599.2   212.3  602.22     222  603.55   270.6  603.74
   280.4  603.98   290.1  604.36   319.3  605.27   338.2  605.66   347.5   606.1
   365.9  608.02   375.1  608.53   384.4  608.78   393.6   608.9     412  608.64
#Mann= 3 , 0 , 0
       0     .08       0   173.3    .045       0   197.3     .06       0
Bank Sta=173.3,197.3
XS Rating Curve= 0 ,0
Exp/Cntr=0.3,0.1

Type RM Length L Ch R = 1 ,2922.5  ,162.3,157.5,152.5
XS GIS Cut Line= 4
     1773685.274      552071.336     1773575.031      551978.454
     1773496.906      551810.919     1773466.524      551733.662
#Sta/Elev= 30
       0  610.13     9.6  609.74    19.2  608.87    38.4  606.56    67.3  603.77
    86.5  602.58    96.1  602.12   124.9  601.27   134.5   601.2   144.2  601.53
   153.9   601.6   163.6  601.41   173.3  600.11   183.1  598.06   192.8  597.07
   202.5  597.46   204.1  597.77   212.3  599.36     222  602.33   231.7  603.75
   241.4  604.14   260.9  603.68   270.6  603.62   299.8  604.01   319.3  603.95
     329  604.18   356.7  605.54   384.4  607.56   393.6  608.06     412  608.58
#Mann= 3 , 0 , 0
       0     .06       0   183.1    .045       0   204.1     .06       0
Bank Sta=183.1,204.1
XS Rating Curve= 0 ,0
Exp/Cntr=0.3,0.1

Type RM Length L Ch R = 1 ,2765    ,137.4,143.7,148.7
XS GIS Cut Line= 4
     1773751.246      552116.475      1773726.94      551923.766
     1773669.649      551849.114     1773596.732      551684.183
#Sta/Elev= 30
       0  611.14     9.7  610.28    19.4  609.78    29.1  609.53    48.6  609.33
    58.3  608.89    87.4  606.99   116.5  604.52   126.2  603.87     136  603.42
   145.7  603.16   184.5  602.51   194.2  601.88   203.6  600.27   213.1   597.9
   222.5  596.72   231.9  596.65   241.3  597.41   250.7  599.26   260.1  600.66
   269.5  601.62   307.3  605.17   316.8  605.71   373.8  607.14   383.2  607.46
   392.7  607.62   402.2  607.44   430.7  605.73   440.2   605.6   468.7  606.24
#Mann= 3 , 0 , 0
       0     .06       0   213.1    .045       0   241.3     .06       0
Bank Sta=213.1,241.3
XS Rating Curve= 0 ,0
Exp/Cntr=0.3,0.1

Type RM Length L Ch R = 1 ,2621.3  ,120.5,121.7,122.4
XS GIS Cut Line= 4
     1773945.473      552139.551      1773931.15      552056.217
     1773728.025       551664.29     1773655.109       551595.28
#Sta/Elev= 30
       0  608.51    28.2  606.62    56.4  603.72    75.2  602.24    94.4  601.24
   133.6  600.41   231.7  600.34   261.1  600.94   300.4  602.31   310.2  602.35
     320  602.06   339.6  600.98   349.4     600   359.2  597.85     369  596.17
   378.8  595.72   388.7  595.86   398.5  596.59   418.1  598.86   437.7  599.99
   467.1  600.38   506.4  602.36     526  603.66   544.2  605.53   562.5  606.86
   580.8  606.42     599  604.88   608.1   604.5   617.3   604.9   626.4  605.68
#Mann= 3 , 0 , 0
       0     .07       0     369    .045       0   398.5     .06       0
Bank Sta=369,398.5
XS Rating Curve= 0 ,0
Exp/Cntr=0.3,0.1

Type RM Length L Ch R = 1 ,2499.6  ,50.9,49,48.6
XS GIS Cut Line= 4
     1774110.621      552081.752     1773893.607      551770.989
     1773810.274      551576.544     1773697.426      551501.891
#Sta/Elev= 30
       0  606.41    19.4  605.88    58.3  604.38    77.8  603.34   106.9  601.23
   116.6  600.73   165.2  599.52   233.2  599.42   359.6  599.89   388.6  599.43
   407.9  599.63   417.5   599.3   427.1  598.28   446.4  595.53   465.6  594.77
   475.2  594.98     478  595.27   484.8  595.97   494.4  597.63     504  598.74
   542.5  601.77   561.7  602.99   571.4   603.2   590.6  602.44   629.2  603.11
   648.6  602.56   667.9  601.46   687.2  601.81   696.9  602.26   725.9  604.32
#Mann= 3 , 0 , 0
       0     .06       0   446.4    .045       0     478     .06       0
Bank Sta=446.4,478
XS Rating Curve= 0 ,0
Exp/Cntr=0.3,0.1

Type RM Length L Ch R = 1 ,2450.6  ,124.7,118.1,111.4
XS GIS Cut Line= 4
     1774150.551      552053.975     1773933.537      551743.211
     1773850.204      551548.766     1773737.357      551474.114
#Sta/Elev= 30
       0  609.93    19.4  608.92    48.6  607.93      68     607    77.8  606.44
   155.5  600.98   165.2  600.39   174.9  600.08   204.1  599.66   252.7   599.3
   330.4   599.2   398.3  599.36   436.7   599.7   446.4  599.19     456   596.8
   463.8  595.18   465.6  594.81   475.2  594.49   484.8  595.12   494.4  596.48
     504  598.07   513.7  598.89   552.1  599.37   571.4  599.14   609.9   599.1
   629.2  599.11   638.9  599.33   658.2  600.76   687.2   603.6   725.9  605.36
#Mann= 3 , 0 , 0
       0     .06       0   463.8    .045       0   484.8     .06       0
Bank Sta=463.8,484.8
XS Rating Curve= 0 ,0
Exp/Cntr=0.3,0.1

Type RM Length L Ch R = 1 ,2332.5  ,55.6,55.6,55.6
XS GIS Cut Line= 6
      1774218.26      551996.683     1774094.996      551823.072
     1774055.065      551696.336     1774029.024      551635.572
     1773926.593      551514.044      1773789.44      551378.627
#Sta/Elev= 30
       0  605.08    19.4  605.15    77.4  604.58    96.8  604.05   154.8  601.73
   212.9  601.39   222.4  601.11   241.4   599.6   269.9  598.97   288.8  599.15
   317.3  600.74   326.8  600.96   364.7  601.03   383.6  600.76   421.3  598.98
   430.6  598.07   447.8     595   458.6  594.14     468  594.31  473.34  595.04
   486.7   596.6     496  597.22   524.1  598.09   552.2  599.83   590.1  600.51
   628.7  600.64   667.2   600.1   705.8  600.55   734.7  601.24   763.6  602.96
#Mann= 3 , 0 , 0
       0     .06       0   447.8    .045       0  473.34     .06       0
Bank Sta=447.8,473.34
XS Rating Curve= 0 ,0
Exp/Cntr=0.3,0.1

Type RM Length L Ch R = 1 ,2276.9  ,56.7,58.4,60.1
XS GIS Cut Line= 6
     1774270.343      551972.377     1774147.079      551798.766
     1774107.149       551672.03     1774081.107      551611.266
     1773978.676      551489.739     1773841.524      551354.322
#Sta/Elev= 30
       0  603.66    38.7  603.59   125.8  602.25   164.5  601.33   231.9   598.7
   336.3  598.38   374.1  597.68   430.6   597.3     440  596.59  456.33  594.36
   458.6  594.12     468   593.9  479.72   594.5   486.7  595.51     496  597.42
   514.8  598.78   524.1  599.89   533.4  601.43   542.8  602.64   552.2  603.22
   570.8  603.14   580.5  602.66   609.4  600.67     619  600.16   628.7  599.95
   647.9  600.39   676.8  602.79   705.8  604.43   715.4  604.69   763.6  603.12
#Mann= 3 , 0 , 0
       0     .06       0  456.33    .045       0  479.72     .06       0
Bank Sta=456.33,479.72
XS Rating Curve= 0 ,0
Exp/Cntr=0.3,0.1

Type RM Length L Ch R = 1 ,2218.5  ,233.8,240.2,246.5
XS GIS Cut Line= 4
     1774362.357      551812.655     1774199.162      551682.447
     1774053.329      551481.058     1773834.579      551238.002
#Sta/Elev= 30
       0  603.14      19  604.63    28.5     605    66.4  605.41   113.9  606.56
   123.4  605.93   151.8  601.91   161.3  601.01     247  598.29   294.8  598.65
   333.1  599.43   342.7  599.25   361.8  597.96   380.9   594.4   390.5  593.61
   399.8  593.71   409.6  594.59   428.7  597.95   447.9  600.22     467  601.89
   495.9   603.3   534.4  603.62   572.8  605.28   601.7  603.66   630.5  603.24
   649.8  603.51   678.6  604.58   736.3  604.14   765.2  605.08   784.4  605.35
#Mann= 3 , 0 , 0
       0     .06       0   380.9    .045       0   409.6     .06       0
Bank Sta=380.9,409.6
XS Rating Curve= 0 ,0
Exp/Cntr=0.3,0.1

Type RM Length L Ch R = 1 ,1978.2  ,404.4,424.6,444
XS GIS Cut Line= 6
     1774407.496      551833.489     1774348.468      551705.016
     1774348.468      551562.655     1774265.135      551323.072
      1774180.04      550982.692     1774078.937      550853.888
#Sta/Elev= 30
       0  599.68      66  602.88    94.3  605.14   141.4  605.24   160.4   603.7
   179.4  600.82   198.3  599.64   283.8  599.22   322.8  597.52   381.3  598.82
   400.8   597.5   410.6  595.82   420.3  593.17   430.1  591.85  442.16  593.14
   459.4  596.82   517.9  599.94   595.9  600.66   634.9  601.74   732.3  607.32
   761.6   607.7   810.3  606.24     859  606.45   907.5  604.15   926.8  604.79
   955.7  608.65   965.3     609     975  608.99  1013.5   606.5    1052  607.16
#Mann= 3 , 0 , 0
       0     .06       0   420.3    .045       0  442.16     .06       0
Bank Sta=420.3,442.16
XS Rating Curve= 0 ,0
Exp/Cntr=0.3,0.1

Type RM Length L Ch R = 1 ,1553.6  ,475.3,477.8,480.6
XS GIS Cut Line= 4
     1774486.923      552186.353     1774479.009      551863.755
     1774796.385      551309.183     1775015.135      551107.794
#Sta/Elev= 30
       0  606.55      88  608.85   215.1  603.22     264  602.04   352.2  601.48
   391.5  603.44     421  603.56     480  599.95   519.3  598.52   597.9   599.4
   656.9   597.4   755.2  596.68   765.1  596.35   774.9  594.12   784.7  591.18
   794.6  590.29   804.4  591.31   814.2  594.47     824  595.46   873.2  595.62
   892.8  596.96     942  597.09   990.4  607.56  1019.2  610.22  1057.6  612.29
  1067.2  614.07  1134.3   641.7  1163.1  650.86  1201.4  661.58    1259  672.61
#Mann= 3 , 0 , 0
       0     .06       0   774.9    .045       0   814.2     .06       0
Bank Sta=774.9,814.2
XS Rating Curve= 0 ,0
Exp/Cntr=0.3,0.1

Type RM Length L Ch R = 1 ,1075.9  ,578,578.4,575.3
XS GIS Cut Line= 4
     1775001.246      552114.739     1775032.496      551774.461
     1775192.218      551562.655     1775279.024      551402.933
#Sta/Elev= 30
       0  599.38    68.3  600.06   126.9  602.41   146.4   602.7   195.3  601.43
   322.2  600.33   371.2  599.05   430.1  598.71     440  598.32   479.3  595.21
   489.1  594.12   498.9  591.78   508.7  589.05   518.6  588.25   528.4  589.66
  533.57  591.73   538.2  594.09     548  598.17   577.5  604.71   587.3  606.46
   597.2  607.64   635.7  609.44   645.3  611.74   654.8  615.76   693.1  635.34
   702.7  639.81   712.2  643.62   750.5  656.79   769.6  664.75   788.8  670.95
#Mann= 3 , 0 , 0
       0     .08       0   498.9    .045       0  533.57     .08       0
Bank Sta=498.9,533.57
XS Rating Curve= 0 ,0
Exp/Cntr=0.3,0.1

Type RM Length L Ch R = 1 ,497.4   ,426.5,405.2,381.6
XS GIS Cut Line= 4
     1775411.402      552035.746     1775420.083      551859.964
      1775530.76      551716.735     1775558.972      551508.402
#Sta/Elev= 30
       0  613.62    48.9  612.41    68.4  613.13      88  614.95     176  613.91
   185.5  612.28     195  608.27   214.1  598.69   223.6  596.81   280.8  594.72
   290.3  593.06   299.8  589.64   309.4  587.49   318.9  587.28   328.4  589.27
     338  596.42   347.5  602.52     357  604.68   404.8  608.88   414.3  611.26
     443  623.16   452.6  626.24   462.1  628.29   471.7  628.84   500.4  628.77
   519.5  630.05     529  633.47   538.6  638.41   548.1  642.35   567.2  647.56
#Mann= 3 , 0 , 0
       0     .08       0   299.8    .045       0   328.4     .08       0
Bank Sta=299.8,328.4
XS Rating Curve= 0 ,0
Exp/Cntr=0.3,0.1

Type RM Length L Ch R = 1 ,92.2    ,86.7,92.2,97.7
XS GIS Cut Line= 3
     1775700.031      552126.891     1775756.454      551883.836
     1775606.715      551495.381
#Sta/Elev= 30
       0  608.27    76.8  604.15   124.8  604.06   153.6  601.43   182.3  600.52
   211.1  597.42   249.5   594.9   259.2   592.8   268.9  589.01   278.6   586.7
   288.2  587.03   297.9   589.5   307.6  595.47   317.3  599.11     356  601.86
   414.1  603.38   452.8  605.08   462.5  605.68   472.2  607.01   481.9  609.39
   501.2  617.48   510.9  620.42   530.3  622.49   559.3  628.68     569  629.59
   598.1  630.85   607.7  632.39   617.4  634.64   646.5  644.71   665.8     650
#Mann= 3 , 0 , 0
       0     .08       0   268.9    .045       0   297.9     .08       0
Bank Sta=268.9,297.9
XS Rating Curve= 0 ,0
Exp/Cntr=0.3,0.1

Chan Stop Cuts=-1
Use User Specified Reach Order=0
Composite Channel Slope=5
